--- GlenFk.prj (project) ---

Proj Title=GlenFk
Current Plan=p01
Default Exp/Contr=0,0
English Units
Geom File=g01
Flow File=f01
Plan File=p01
BEGIN DESCRIPTION:
END DESCRIPTION:
DSS Export Rating Curves= 0
DSS Export Rating Curve Sorted= 0
DSS Export Volume Flow Curves= 0
DXF OffsetX= 0
DXF OffsetY= 0
DXF ScaleX= 0
DXF ScaleY= 0

--- GlenFk.p01 (plan) ---

Plan Title=Floodplain
Program Version=4.00
Geom File=g01
Flow File=f01
K Sum by GR=0
Std Step Tol=0.01
Critical Tol=0.01
Num of Std Step Trials=20
Max Error Tol=0.3
Flow Tol Ratio=0.001
Split Flow NTrial=30
Split Flow Tol=0.02
Split Flow Ratio=0.02
Log Output Level=0
Friction Slope Method=1
Unsteady Friction Slope Method=2
Unsteady Bridges Friction Slope Method=1
Global Log Level=0
CheckData=False
Run HTab=0
Run UNet=0
Run PostProcess=0
UNET Theta=0
UNET Theta Warmup=0
UNET ZTol=0
UNET ZSATol=0
UNET MxIter=0
UNET MaxInSteps=0
UNET DtIC=0
UNET DtMin=0
UNET MaxCRTS=0
UNET WFStab=0
UNET SFStab=0
UNET WFX=0
UNET SFX=0
UNET DSS MLevel=0
UNET DZMax Abort=0
UNET Convert EG Bridges=0
UNET Use Existing IB Tables=0
UNET Froude Limit=0
UNET Froude Power=0
Write IC File=0
Echo Input=False
Echo Output=False
Write Detailed=0

--- GlenFk.f01 (steady flow) ---

Flow Title=NFF Regression Equation
Program Version=4.00
Number of Profiles=1
Profile Names=P100yr
River Rch & RM=GlenFk,Main      ,14728.3
607.5859
River Rch & RM=GlenFk,Main      ,14400.4
630.3809
River Rch & RM=GlenFk,Main      ,12585.3
685.9554
River Rch & RM=GlenFk,Main      ,12305
776.6137
River Rch & RM=GlenFk,Main      ,11632.2
812.7718
River Rch & RM=GlenFk,Main      ,9220.8
864.0924
River Rch & RM=GlenFk,Main      ,8884.1
959.2371
River Rch & RM=GlenFk,Main      ,6456.4
1049.814
River Rch & RM=GlenFk,Main      ,4969.6
1139.483
River Rch & RM=GlenFk,Main      ,2924.3
1182.238
River Rch & RM=GlenFk,Main      ,2562
1575.728
River Rch & RM=GlenFk,Main      ,160.5
1621.366
Boundary for River Rch & Prof#=GlenFk,Main      ,1
Up Type=0
Dn Type=3
Dn Slope=0.044279

--- GlenFk.g01 (geometry) ---

Geom Title=USGS 10m DEM
Program Version=4.00

River Reach=GlenFk          ,Main
Reach XY= 30
     1825575.533      261127.865      1824485.24      259474.725
     1824514.773      259174.252      1824280.64       258771.63
     1824351.755      258549.532     1824225.936      258386.514
     1824255.114        258107.3     1824070.618      257887.268
     1824088.764      257630.198     1823957.887      257120.664
     1823493.997      256135.992     1823078.024       256020.03
     1822684.378      255750.877     1822239.672      255675.253
     1821936.028      255326.374     1821713.929      255251.976
     1820497.642      255447.822     1819899.945       255687.42
     1819762.091      255475.169     1819449.185      255316.527
     1819244.669      255423.043     1818863.905      255342.032
     1818077.209      254959.857     1817910.002      254658.464
     1817427.314      254209.649     1817182.947        253855.8
     1816918.618      253797.127     1816781.312      253889.672
       1816345.2      253675.548      1815915.11      253800.013

Type RM Length L Ch R = 1 ,14728.3 ,330,327.9,325.8
XS GIS Cut Line= 3
     1826010.347      260963.931      1825577.32      261103.616
     1825144.292      261243.302
#Sta/Elev= 30
       0 1885.89      10 1882.72      50 1865.34      65 1860.91     120 1841.44
     150 1832.14     185 1823.38     210 1818.25     255 1802.73     330 1767.63
     370 1747.14     415 1718.37     425 1710.37     440 1695.59     445 1691.96
     459 1685.28   464.9 1683.88     474 1684.45   519.3 1686.93     544 1686.86
   573.7 1688.12     633 1691.36   677.6 1694.78   766.6 1699.08   781.4  1703.1
   840.8 1724.56   875.4 1740.09   880.3 1741.57   890.2  1738.8     910 1745.16
#Mann= 3 , 0 , 0
       0      .1       0     459    .045       0     474      .1       0
Bank Sta=459,474
XS Rating Curve= 0 ,0
Exp/Cntr=0.3,0.1

Type RM Length L Ch R = 1 ,14400.4 ,348.7,346.8,344.9
XS GIS Cut Line= 4
     1825852.839       260586.48     1825518.719      260784.436
     1825415.324      260826.638     1825035.953       260988.19
#Sta/Elev= 30
       0  1845.3    24.9 1842.15    49.8 1834.83    99.6 1824.26   119.5 1822.52
   159.3 1816.43   189.2 1808.58   209.1 1799.76   288.8 1757.41   313.7 1748.89
   338.6 1741.92   343.6  1739.5   388.4 1711.99   427.2 1686.24   432.1 1683.91
   446.6 1679.79   461.2 1677.38   514.9 1677.24   541.9 1677.63   556.9 1678.08
   589.5 1678.33   614.3 1680.27     659 1695.95   708.7 1723.28   723.6 1729.58
   738.5  1737.7   803.1 1776.62     813 1783.73   862.7 1814.44   912.4  1842.4
#Mann= 3 , 0 , 0
       0      .1       0   541.9    .045       0   556.9      .1       0
Bank Sta=541.9,556.9
XS Rating Curve= 0 ,0
Exp/Cntr=0.3,0.1

Type RM Length L Ch R = 1 ,14053.7 ,762.3,770.2,778.2
XS GIS Cut Line= 4
     1825648.341      260227.462     1825309.818       260467.92
     1825231.744      260527.003     1824878.254      260713.885
#Sta/Elev= 30
       0 1869.99    24.7 1858.36    54.4 1852.82   128.5 1820.26   158.2 1809.91
   197.7  1803.7   237.3 1795.54   271.9 1784.81   331.2 1761.94   370.7 1736.87
   385.6 1726.13   415.2 1711.17   449.5 1679.65   459.3 1671.87     474 1667.93
   498.5 1672.07   543.1 1672.47   558.1 1672.27   558.1 1672.26   578.1 1673.12
   588.1 1675.34   613.1 1689.24   648.1 1701.21   713.1 1730.73     753  1755.1
     788 1773.78     828 1800.89     863 1820.84     888 1839.55     913    1855
#Mann= 3 , 0 , 0
       0      .1       0   543.1    .045       0   558.1      .1       0
Bank Sta=543.1,558.1
XS Rating Curve= 0 ,0
Exp/Cntr=0.3,0.1

Type RM Length L Ch R = 1 ,13283.5 ,488.2,475.1,461.8
XS GIS Cut Line= 4
     1825254.956      259562.685     1824983.789      259800.664
     1824845.595      259887.641     1824472.811      259948.857
#Sta/Elev= 30
       0 1885.46    24.7 1884.98    44.5 1882.18    69.2 1876.74      84 1874.87
   108.7 1866.53   143.3 1846.49   207.6 1805.38   266.9 1770.72   301.5 1747.92
   336.1 1727.34   365.7 1705.77   395.4 1677.55   405.3 1669.18   415.2 1663.23
   430.1  1656.4     440 1653.34   582.7 1651.64   597.7 1651.48   603.6 1651.39
   623.5 1651.74   653.3 1655.68   668.2 1661.73     708 1684.82     713 1686.68
   732.8 1688.79   742.8 1692.51   767.6 1708.57   812.4 1733.48   901.8 1790.29
#Mann= 3 , 0 , 0
       0      .1       0   582.7    .045       0   597.7      .1       0
Bank Sta=582.7,597.7
XS Rating Curve= 0 ,0
Exp/Cntr=0.3,0.1

Type RM Length L Ch R = 1 ,12808.4 ,205.9,223.1,240.3
XS GIS Cut Line= 4
      1825149.45      259431.858     1824693.667      259419.198
     1824533.299      259488.831     1824268.811      259718.872
#Sta/Elev= 30
       0 1796.43    24.8 1787.24    74.3 1772.02   123.9 1759.19     228 1735.79
   267.6 1722.44   312.2 1710.43   327.1 1707.22     342 1705.89   376.7 1697.18
   386.6  1692.9     446 1660.93   500.9 1641.65   545.9 1643.46   600.8  1640.6
   659.9 1640.98   674.9  1640.4   675.2 1640.39   729.5 1643.37   744.3 1646.36
   764.1 1653.34     774 1659.59   798.6 1684.43   818.4 1699.34   833.2 1708.94
   857.9 1720.04   872.7 1729.37   887.5 1741.11   941.8 1762.71   981.3 1773.75
#Mann= 3 , 0 , 0
       0      .1       0   659.9    .045       0   674.9      .1       0
Bank Sta=659.9,674.9
XS Rating Curve= 0 ,0
Exp/Cntr=0.3,0.1

Type RM Length L Ch R = 1 ,12585.3 ,287.5,280.2,272.9
XS GIS Cut Line= 4
     1824989.082      259163.875     1824575.502      259303.142
     1824451.005      259298.922     1824191.462       259467.73
#Sta/Elev= 30
       0 1767.72    44.6 1753.36    69.4 1746.48    79.4 1742.66   128.9 1731.28
   138.8 1728.45   173.6 1714.99   203.3 1700.61   208.3 1699.39   233.1 1702.33
     243 1701.85   252.9 1700.43   327.3 1680.39   347.1 1675.94   396.7 1653.41
   401.7 1651.82   421.5 1651.97   436.4 1650.94   471.3 1639.78   487.5 1638.43
   502.5 1637.71   511.1  1637.5   635.9 1641.21   680.8 1644.63   695.8 1646.87
   715.8 1648.43   750.7 1649.76   785.7 1649.47   815.6    1652   870.6 1655.23
#Mann= 3 , 0 , 0
       0      .1       0   487.5    .045       0   502.5      .1       0
Bank Sta=487.5,502.5
XS Rating Curve= 0 ,0
Exp/Cntr=0.3,0.1

Type RM Length L Ch R = 1 ,12305   ,208.3,207.6,206.8
XS GIS Cut Line= 4
     1824921.443      258847.996     1824592.382      258992.956
     1824309.628      259077.361     1824031.622       259045.58
#Sta/Elev= 30
       0  1920.4      30 1896.92      45 1886.68    59.9 1872.26    64.9 1868.79
    79.9 1862.22    89.9 1860.73    99.9 1856.61   124.8 1837.75   159.8  1818.6
   279.7 1745.43   349.6 1712.17     394 1688.87   428.4 1661.48   448.1 1647.49
   457.9 1641.75   477.6 1634.07   493.5 1633.87   508.5 1633.49   590.7 1633.03
   620.2  1633.5   659.7 1636.98   679.6 1640.52   694.6  1647.4   719.6 1648.73
   729.6 1650.47   744.6 1662.68   844.5 1713.21   899.5 1743.93   934.5 1758.64
#Mann= 3 , 0 , 0
       0      .1       0   493.5    .045       0   508.5      .1       0
Bank Sta=493.5,508.5
XS Rating Curve= 0 ,0
Exp/Cntr=0.3,0.1

Type RM Length L Ch R = 1 ,12097.5 ,468.9,465.3,461.6
XS GIS Cut Line= 4
     1824822.384      258632.128      1824539.63      258803.047
     1824221.004      258908.552     1823997.333      258885.341
#Sta/Elev= 30
       0 1864.59    29.6 1862.24    44.4 1858.84      69 1855.82    93.7  1849.1
   113.4 1840.26   123.3 1837.95   138.1 1837.08   147.9 1832.94   162.7 1824.64
   197.2 1802.39   300.8 1728.21   355.1 1696.38   404.4 1652.81   429.1 1635.19
   448.9 1632.33   542.7  1630.2   552.5 1629.76   557.7 1629.93   567.3 1631.23
   587.1 1631.05   611.7 1634.63   631.5 1648.09   636.4  1650.4   651.2  1654.2
     666 1661.95     676 1665.75     706 1673.79     811 1713.94   890.9 1755.02
#Mann= 3 , 0 , 0
       0      .1       0   542.7    .045       0   557.7      .1       0
Bank Sta=542.7,557.7
XS Rating Curve= 0 ,0
Exp/Cntr=0.3,0.1

Type RM Length L Ch R = 1 ,11632.2 ,429.5,431.6,433.8
XS GIS Cut Line= 3
     1824738.694      258273.592      1824349.72      258429.558
      1823895.13      258654.051
#Sta/Elev= 30
       0 1733.71    39.9 1722.21   134.7 1691.88   169.6 1689.75   209.5 1683.59
   274.4 1668.85   294.4  1661.6   329.3 1655.78   344.2 1655.34   359.2 1652.37
   389.1 1649.55   409.1 1643.51   443.9 1638.17   448.9 1636.24   463.8 1627.48
   471.8 1624.18   478.7 1622.76   486.8 1623.56   523.5 1628.07   553.3 1629.69
   573.2 1634.89   588.1 1636.45   622.9 1643.84   657.7  1649.3   692.5 1658.57
   707.4 1661.41   722.3  1665.7   801.8  1696.6   826.7    1704   926.1 1738.49
#Mann= 3 , 0 , 0
       0      .1       0   471.8    .045       0   486.8      .1       0
Bank Sta=471.8,486.8
XS Rating Curve= 0 ,0
Exp/Cntr=0.3,0.1

Type RM Length L Ch R = 1 ,11200.5 ,560.6,564.1,567.6
XS GIS Cut Line= 4
     1824576.237      257748.443     1824375.042      258037.078
     1824079.627      258136.253     1823798.564      258269.334
#Sta/Elev= 30
       0 1833.99    24.8 1827.45    44.6 1817.16   104.1    1796   153.6 1776.13
   183.4  1762.6   203.2 1751.47     223 1741.99   282.5  1719.3     337 1695.56
     426 1650.55   460.7 1635.21   483.1 1623.81   490.3 1620.77   495.3 1619.93
   498.1 1620.09   529.9 1623.26     614 1622.08   638.7 1622.98   683.2 1640.18
     703 1646.87   747.4 1670.02     777 1687.89   796.7 1698.47   831.3 1723.11
     856 1738.93   880.6 1757.54     930  1792.2   944.8 1799.93   974.4 1820.86
#Mann= 3 , 0 , 0
       0      .1       0   483.1    .045       0   498.1      .1       0
Bank Sta=483.1,498.1
XS Rating Curve= 0 ,0
Exp/Cntr=0.3,0.1

Type RM Length L Ch R = 1 ,10636.5 ,473.3,473,472.6
XS GIS Cut Line= 3
     1824525.523      257505.562     1824193.573      257577.076
     1823618.991       257684.47
#Sta/Elev= 30
       0 1862.88      30 1836.91    44.9  1831.4    54.9 1826.24    84.9 1801.49
   119.8 1776.72   164.8 1747.46   219.7 1714.73   264.7    1690   334.6 1655.12
   349.6 1649.99   399.5 1629.55   424.5 1617.57   444.7 1613.14   449.5  1612.9
   459.7 1613.68   524.4 1614.95   534.4 1617.64   554.4 1628.18   559.4 1629.98
   589.4 1633.28   599.4 1635.57   624.3 1647.29   684.3 1671.93   714.3 1685.67
   734.2 1696.69   769.2 1714.14   814.2 1733.64   889.1 1773.28   924.1 1796.35
#Mann= 3 , 0 , 0
       0      .1       0   444.7    .045       0   459.7      .1       0
Bank Sta=444.7,459.7
XS Rating Curve= 0 ,0
Exp/Cntr=0.3,0.1

Type RM Length L Ch R = 1 ,10163.5 ,342.8,339.7,336.5
XS GIS Cut Line= 4
     1824305.408       256874.41     1824014.214      257146.614
     1823906.598      257167.715     1823481.519       257200.08
#Sta/Elev= 30
       0  1767.6    19.9 1756.56    49.8    1743    99.6 1716.87   139.5 1694.01
   184.4  1670.4   239.2 1638.63     279 1631.46   353.8 1622.82   398.6 1614.29
   418.6 1609.17   442.9 1604.45   448.5 1604.09   457.9 1604.67   493.3 1606.81
   523.1    1607   547.9 1609.02   582.6 1614.83   602.5  1616.6   632.2 1628.13
   661.9 1632.68   701.6 1633.42   706.6 1635.08   736.3 1647.91   761.1 1661.32
   795.8 1684.77   840.4 1717.28     890 1749.52   909.8 1764.11   934.6 1779.86
#Mann= 3 , 0 , 0
       0      .1       0   442.9    .045       0   457.9      .1       0
Bank Sta=442.9,457.9
XS Rating Curve= 0 ,0
Exp/Cntr=0.3,0.1

Type RM Length L Ch R = 1 ,9823.9  ,180,180.2,180.4
XS GIS Cut Line= 4
     1824237.885      256756.245     1823879.167      256827.988
     1823782.102       256861.75     1823461.366      257102.302
#Sta/Elev= 30
       0 1791.27    34.6 1774.99    59.3 1761.36    79.1 1751.35   113.7 1739.29
   143.4 1726.25   187.8 1701.55   202.7    1694   247.2 1668.36   271.9  1652.9
   311.4 1631.57   375.6 1601.74   380.5 1600.55   398.9 1598.68     405 1598.39
   413.9 1598.73   434.3 1600.12     449  1600.1   453.9 1601.32   488.4 1617.19
   597.3 1654.44   612.1 1660.18   646.8 1675.33   671.5 1687.61     721  1714.5
   765.6 1736.73   795.3 1754.01     820 1769.51   839.8  1780.7   869.5 1799.66
#Mann= 3 , 0 , 0
       0      .1       0   398.9    .045       0   413.9      .1       0
Bank Sta=398.9,413.9
XS Rating Curve= 0 ,0
Exp/Cntr=0.3,0.1

Type RM Length L Ch R = 1 ,9643.7  ,426.6,422.9,419.2
XS GIS Cut Line= 3
     1824188.327       256501.86     1823849.625      256648.629
     1823335.996      256822.538
#Sta/Elev= 30
       0 1769.22    29.9 1750.94    69.8 1733.37    89.8 1723.48   134.7 1698.55
   194.5 1670.72   214.5 1664.18   254.4 1653.65   284.3 1641.23   324.2 1631.88
   349.2 1624.66   384.1 1611.12   418.9 1605.51   438.5 1598.13   448.7 1594.65
   453.5 1595.15   473.6 1597.89   483.6 1601.21   508.4 1614.79   573.1 1645.43
   627.8 1673.07   657.7 1690.09   687.5 1709.45   722.4 1728.68   752.2 1746.54
   767.1 1756.29     802 1777.23   846.7 1806.63   886.5 1831.85   911.4 1846.63
#Mann= 3 , 0 , 0
       0      .1       0   438.5    .045       0   453.5      .1       0
Bank Sta=438.5,453.5
XS Rating Curve= 0 ,0
Exp/Cntr=0.3,0.1

Type RM Length L Ch R = 1 ,9220.8  ,355.2,336.7,318.3
XS GIS Cut Line= 4
     1824005.773      256159.085     1823644.945       256268.81
     1823526.779      256332.113     1823219.714      256573.047
#Sta/Elev= 30
       0 1674.81    24.8  1671.7    74.4    1668   104.2 1664.81   153.8 1657.71
   188.6 1651.52     258 1625.87   272.9 1621.31   292.8 1618.41   312.6 1614.38
   347.4 1602.67   387.1 1598.96     402 1594.75   415.7 1589.46   421.8 1588.16
   426.8 1588.09   430.7 1588.51   451.6 1592.34   471.5 1593.05   476.4 1594.57
   555.7 1632.51   600.1  1650.5     615  1657.3   708.8 1704.01   723.6 1710.48
   758.2 1722.46   782.9 1733.33   812.6 1744.21     862 1768.44   901.5 1790.45
#Mann= 3 , 0 , 0
       0      .1       0   415.7    .045       0   430.7      .1       0
Bank Sta=415.7,430.7
XS Rating Curve= 0 ,0
Exp/Cntr=0.3,0.1

Type RM Length L Ch R = 1 ,8884.1  ,80.2,84.2,88.2
XS GIS Cut Line= 4
     1823638.615      255829.908     1823368.521       256066.24
       1823343.2      256159.085      1823138.52      256522.023
#Sta/Elev= 30
       0  1752.9    34.9 1742.92    64.8 1732.68   104.7 1717.43   164.5 1685.61
   184.4 1673.06   219.3 1655.49   279.1 1619.68   289.1 1615.13     334 1600.27
   363.7 1582.69   368.5  1580.4   377.8 1578.82   392.8 1576.26   402.2  1575.1
   411.8 1576.52   431.1 1587.02   440.7  1590.9   460.1  1590.9   494.8 1601.67
   519.6 1607.02   539.4 1612.54   574.2 1625.74   608.9 1640.84   658.5 1666.02
     718    1700   752.8 1717.44   772.6 1728.35   817.2 1756.16   871.8 1788.03
#Mann= 3 , 0 , 0
       0      .1       0   377.8    .045       0   392.8      .1       0
Bank Sta=377.8,392.8
XS Rating Curve= 0 ,0
Exp/Cntr=0.3,0.1

Type RM Length L Ch R = 1 ,8799.9  ,178.2,173.3,168.4
XS GIS Cut Line= 4
     1823425.494      255707.522     1823290.447      256053.579
     1823244.025      256156.974     1823043.565       256467.16
#Sta/Elev= 30
       0 1736.87    74.3 1713.02   128.8 1690.22   153.5 1678.86   188.2 1661.34
     213 1654.09   237.7 1644.22   252.6 1636.35   292.2 1612.22   302.1 1608.38
   336.8 1599.46   356.6 1587.39   366.5 1582.68   376.4 1579.58   393.9 1576.71
     406 1575.56   408.9 1575.77   415.8 1576.87   440.5 1584.86   465.1 1585.15
   484.8 1593.38   499.8 1597.25   519.8 1605.63   554.7 1623.47   579.6 1637.34
   634.5    1673   664.5 1690.83   769.3 1749.39   794.2 1761.57   854.1 1785.61
#Mann= 3 , 0 , 0
       0      .1       0   393.9    .045       0   408.9      .1       0
Bank Sta=393.9,408.9
XS Rating Curve= 0 ,0
Exp/Cntr=0.3,0.1

Type RM Length L Ch R = 1 ,8626.6  ,463.9,469.6,475.3
XS GIS Cut Line= 4
     1823241.757       255583.65     1823127.969      255969.175
     1823100.538      256087.341     1822927.509      256435.508
#Sta/Elev= 30
       0 1720.55    74.4 1682.52   119.1 1660.33     129 1655.92     139 1652.65
   168.7 1640.59   188.6 1629.74   203.5 1623.29   213.4  1621.4   238.2 1618.78
   253.1 1615.96   272.9 1610.71   302.7  1601.2   357.3 1589.23   377.2 1582.91
   406.8 1578.44   431.1  1577.8   457.2 1572.47     465 1570.55   472.2 1571.21
   484.5 1574.46   533.2 1590.56   563.2 1599.12     603 1612.72     618 1618.49
   677.8 1645.78   717.7 1665.54   762.5 1684.31   877.2 1735.46   912.1 1753.27
#Mann= 3 , 0 , 0
       0      .1       0   457.2    .045       0   472.2      .1       0
Bank Sta=457.2,472.2
XS Rating Curve= 0 ,0
Exp/Cntr=0.3,0.1

Type RM Length L Ch R = 1 ,8157    ,554.4,561.2,568
XS GIS Cut Line= 4
     1822902.104      255365.872      1822750.26      255726.513
     1822693.288      255836.238     1822472.628      256168.787
#Sta/Elev= 30
       0 1654.17    29.7 1636.15    39.6 1632.25    84.2 1629.25     104 1626.64
   123.8 1621.06   148.6 1610.52   178.3 1602.38   222.9 1596.96   257.6 1590.38
   272.4 1588.82   307.1  1583.3   336.8 1581.36   361.6 1575.66   406.1 1563.02
   434.7 1558.31   440.8 1557.38   449.7 1558.92   470.4  1562.1     505 1564.24
     510 1565.34   524.9  1569.9   549.9 1580.59   684.6 1630.45   704.5 1636.36
   744.4 1640.79   769.4 1646.01   789.3 1643.57   839.2 1632.53     914 1620.34
#Mann= 3 , 0 , 0
       0      .1       0   434.7    .045       0   449.7      .1       0
Bank Sta=434.7,449.7
XS Rating Curve= 0 ,0
Exp/Cntr=0.3,0.1

Type RM Length L Ch R = 1 ,7595.7  ,138.6,138.9,139.2
XS GIS Cut Line= 4
     1822443.671       255210.71     1822243.835      255602.017
     1822159.431      255686.421     1822003.359      256054.627
#Sta/Elev= 30
       0 1668.52      15  1661.7    49.9 1643.54    89.9 1625.24   164.8 1597.62
   189.7 1589.77   249.6 1578.86   284.6 1571.25   339.5 1554.88   359.5  1550.4
   369.5  1549.4   414.4 1550.51   469.2 1549.19   494.1 1545.66     499 1545.82
     514 1548.97     514 1548.98   523.9 1552.26   528.9 1554.84   558.8  1573.5
   593.7    1591   703.7 1663.22   753.7 1692.12   783.7 1711.81   808.7 1726.78
   843.7 1746.52   873.7 1760.37   903.7 1771.18   933.7 1777.53   958.7 1781.31
#Mann= 3 , 0 , 0
       0      .1       0     499    .045       0     514      .1       0
Bank Sta=499,514
XS Rating Curve= 0 ,0
Exp/Cntr=0.3,0.1

Type RM Length L Ch R = 1 ,7456.9  ,130.9,138.8,146.8
XS GIS Cut Line= 4
      1822343.01      255194.766     1822218.514      255433.208
     1822037.045      255614.677     1821931.539      255960.735
#Sta/Elev= 30
       0 1635.97    24.9  1627.7    99.6 1607.07   224.2 1565.53   244.1 1560.46
   278.9 1549.65   288.7 1548.04   313.4 1546.29   338.1 1546.68   352.9 1545.48
   372.6 1545.97   407.2 1541.28   415.3 1542.13   430.3 1545.01   436.8 1547.18
   446.7 1552.19   466.4 1563.82   505.9 1585.47   525.6 1596.91   540.5 1604.11
   555.4 1612.22   575.2 1623.36   614.8 1648.24   679.3    1684     709  1701.6
   763.5 1736.16   783.3 1749.59   813.1 1767.81   832.9 1780.98   887.4 1812.61
#Mann= 3 , 0 , 0
       0      .1       0   415.3    .045       0   430.3      .1       0
Bank Sta=415.3,430.3
XS Rating Curve= 0 ,0
Exp/Cntr=0.3,0.1

Type RM Length L Ch R = 1 ,7318    ,373.2,359.5,337.9
XS GIS Cut Line= 4
     1822292.367      255158.895     1822155.211      255372.015
     1821954.751       255464.86     1821826.034      255893.211
#Sta/Elev= 30
       0 1623.72    39.8 1614.45    69.6 1608.92   119.3 1593.29     159 1582.55
   203.8 1568.37   233.6 1558.09   258.4 1547.54   263.3 1546.13   268.2 1545.32
   282.9 1544.96   356.5 1544.29   389.2 1544.56   404.2 1544.55   420.4 1544.47
   425.3 1545.45   444.9 1551.28   474.4 1562.15   514.1 1580.19   548.9 1595.13
   608.5 1622.54   643.3  1641.5   658.2 1650.38   717.9 1681.97   762.6 1712.82
   827.2 1752.89   852.1  1769.2   871.9 1783.01   906.7 1805.15   921.6 1813.93
#Mann= 3 , 0 , 0
       0      .1       0   389.2    .045       0   404.2      .1       0
Bank Sta=389.2,404.2
XS Rating Curve= 0 ,0
Exp/Cntr=0.3,0.1

Type RM Length L Ch R = 1 ,6958.5  ,318.9,310.3,309.1
XS GIS Cut Line= 3
     1822022.597      254901.545      1821737.41      255245.409
     1821662.663      255747.825
#Sta/Elev= 30
       0 1706.54    44.7 1699.75    69.5 1692.55    89.4 1684.02   124.1 1672.02
   183.7 1643.87   203.5 1633.29     268 1603.72   287.9 1597.03   322.6 1581.17
   357.4 1570.47   377.2  1563.3     417 1546.46   441.8 1534.27   448.8 1532.15
   451.7 1532.12   463.8 1534.72   486.6 1537.94   536.4 1537.56   561.3 1539.48
   566.2 1541.01   591.2  1551.5     626 1568.89   675.8 1597.66   745.5 1636.22
   765.4 1646.28   810.3  1666.2     865 1695.36   904.9 1711.65   954.7 1734.68
#Mann= 3 , 0 , 0
       0      .1       0   448.8    .045       0   463.8      .1       0
Bank Sta=448.8,463.8
XS Rating Curve= 0 ,0
Exp/Cntr=0.3,0.1

Type RM Length L Ch R = 1 ,6648.2  ,199.9,191.8,184.2
XS GIS Cut Line= 3
     1821355.084      254809.721     1821433.555      255213.757
     1821408.435      255719.173
#Sta/Elev= 30
       0 1641.46    59.5 1631.58    99.2 1622.05   128.9 1613.48   183.5 1607.42
   208.3 1602.32   257.9  1589.1   292.6 1576.95   312.4 1568.92   342.2 1561.65
     367 1554.03   421.5 1533.19   431.4 1530.71   443.5 1528.84   458.5 1527.95
   461.2 1527.93   471.1 1528.41     486 1530.44   520.7 1537.38   595.2 1549.13
   605.1 1551.83     620 1558.86   644.8  1568.6   679.5 1590.15   704.3 1602.93
   734.1 1620.17   763.8 1635.66   848.2 1673.19   887.9 1692.45   917.6 1708.55
#Mann= 3 , 0 , 0
       0      .1       0   443.5    .045       0   458.5      .1       0
Bank Sta=443.5,458.5
XS Rating Curve= 0 ,0
Exp/Cntr=0.3,0.1

Type RM Length L Ch R = 1 ,6456.4  ,721.8,724.8,727.7
XS GIS Cut Line= 4
     1821161.272      254874.014     1821233.094      255239.079
     1821271.076      255395.226     1821322.395      255776.919
#Sta/Elev= 30
       0 1668.38    64.5 1647.89   119.1 1631.82   153.8 1618.56   183.6 1604.93
   203.4 1596.91   277.8 1571.38   322.4 1550.17   332.4 1547.25   352.2 1545.44
   396.4 1527.55   410.8 1522.66   415.9 1521.94   425.8 1523.31   474.3 1525.58
   488.9 1525.53   498.7 1526.55   508.4 1528.23   547.6 1538.03   572.3 1543.01
   616.7 1562.48   641.4 1575.12     676 1589.02   705.6 1603.23   730.3 1611.92
     755 1618.84   769.8 1625.11   838.9 1669.32   868.5 1685.21   917.9 1714.68
#Mann= 3 , 0 , 0
       0      .1       0   410.8    .045       0   425.8      .1       0
Bank Sta=410.8,425.8
XS Rating Curve= 0 ,0
Exp/Cntr=0.3,0.1

Type RM Length L Ch R = 1 ,5731.7  ,479.3,472.2,465.1
XS GIS Cut Line= 4
     1820642.265      255023.848      1820543.09      255342.474
     1820566.301      255553.484     1820728.779      255888.991
#Sta/Elev= 30
       0 1654.45   219.2 1576.78   239.1 1570.47     264 1563.94   303.8 1550.17
   323.7 1544.07   333.7 1539.72   363.3 1523.33     388 1510.84   425.4 1505.51
   432.4 1504.95   440.4 1505.73   496.6 1511.36   501.6 1513.16   511.4 1518.07
     541 1528.98   560.9 1537.12   610.6 1558.49   640.4  1573.4   670.2 1589.66
     705 1616.27     710 1619.58     715 1622.18   729.9 1627.72   769.6 1647.82
   799.5 1663.76   819.4 1676.06   859.1 1696.51   898.9 1715.25   918.8 1721.37
#Mann= 3 , 0 , 0
       0      .1       0   425.4    .045       0   440.4      .1       0
Bank Sta=425.4,440.4
XS Rating Curve= 0 ,0
Exp/Cntr=0.3,0.1

Type RM Length L Ch R = 1 ,5259.5  ,137.3,143.9,150.6
XS GIS Cut Line= 4
     1820116.849      255129.353     1820097.858      255566.145
     1820180.152      255747.614     1820424.924      255935.413
#Sta/Elev= 30
       0 1770.35    19.9 1762.08    64.6 1729.95    99.4 1707.76   134.1 1683.24
   193.8 1646.77   268.3 1596.42     308 1566.34   342.8 1544.97   377.6 1527.55
   412.4 1514.89   437.2 1499.82   442.2 1497.96   490.1 1496.59     497 1496.43
   505.1 1496.64   536.8 1499.08   621.5  1500.5   631.5 1501.28   641.4 1503.29
   666.3 1510.86   691.2 1520.87     726 1532.65   745.9 1540.48   790.7 1555.03
   830.5 1571.42   875.3 1585.42   885.3  1588.1   900.2 1590.46     945 1593.34
#Mann= 3 , 0 , 0
       0      .1       0   490.1    .045       0   505.1      .1       0
Bank Sta=490.1,505.1
XS Rating Curve= 0 ,0
Exp/Cntr=0.3,0.1

Type RM Length L Ch R = 1 ,5115.5  ,120,146,171.9
XS GIS Cut Line= 4
     1820056.096      255086.383     1819990.242      255648.439
     1820000.793      255728.623     1820058.261      256081.067
#Sta/Elev= 30
       0 1759.13    14.9 1757.99    24.8 1755.05    54.6 1744.16    84.4 1730.35
   153.9 1689.42   173.7 1676.42   183.7 1670.64   228.4 1647.62   258.1 1633.44
     278 1615.52   297.8 1600.65   312.7 1591.39   332.6 1580.33   387.2 1542.64
     412 1533.43   431.9 1524.92   476.6 1499.98   481.5 1498.43   506.3 1496.65
     546  1494.5   570.7 1494.37     595  1494.8     610 1495.45   701.3 1499.27
   731.1 1503.48   820.4  1518.2   904.7 1539.24   964.2 1550.21  1003.9 1556.66
#Mann= 3 , 0 , 0
       0      .1       0     595    .045       0     610      .1       0
Bank Sta=595,610
XS Rating Curve= 0 ,0
Exp/Cntr=0.3,0.1

Type RM Length L Ch R = 1 ,4969.6  ,391.8,381.8,371.9
XS GIS Cut Line= 4
      1819950.15      255112.472     1819901.618      255633.668
     1819808.773      255692.751     1819760.241      256000.827
#Sta/Elev= 30
       0  1686.6    19.9 1682.07    89.7 1659.43   134.6 1648.55   144.6 1645.15
   184.4 1622.99   209.4  1612.2   249.3 1591.98   269.2 1578.63   309.1 1549.34
     349 1533.09   363.9 1525.89   388.8 1518.85   423.8 1497.97   468.6 1489.32
   566.7 1488.57   580.9 1485.85   581.7 1485.93   585.6 1486.32   590.4 1488.32
   623.9 1505.83   653.3 1508.74     678  1512.5   712.7 1524.85   732.5 1532.87
   757.3 1544.78   791.9 1563.04   816.7 1570.74   915.7 1605.52   945.4 1618.05
#Mann= 3 , 0 , 0
       0      .1       0   566.7    .045       0   581.7      .1       0
Bank Sta=566.7,581.7
XS Rating Curve= 0 ,0
Exp/Cntr=0.3,0.1

Type RM Length L Ch R = 1 ,4587.7  ,135.4,122.8,110.2
XS GIS Cut Line= 4
     1819843.544      254994.221     1819658.956      255346.694
     1819580.882       255458.53     1819415.406      255878.351
#Sta/Elev= 30
       0 1605.18    24.9 1598.88    64.7 1592.48   134.3 1578.48     194 1564.08
   208.9 1559.44   218.8 1554.96   243.7    1546   273.5 1537.17   323.3 1516.84
   363.1 1499.39     383 1491.93   387.9 1490.47   412.5 1487.07   451.5 1476.87
   461.2 1476.02   466.5 1476.84   490.4 1481.43   539.2 1482.98   559.1 1485.05
     569 1487.03   613.6 1503.99   648.3 1513.06     688 1528.24   742.6 1546.49
   772.3 1559.95     802 1576.85   831.8  1590.8   856.6 1604.79   985.5  1685.2
#Mann= 3 , 0 , 0
       0      .1       0   451.5    .045       0   466.5      .1       0
Bank Sta=451.5,466.5
XS Rating Curve= 0 ,0
Exp/Cntr=0.3,0.1

Type RM Length L Ch R = 1 ,4464.9  ,459.7,465.8,472
XS GIS Cut Line= 4
     1819614.644      254983.756     1819515.469      255298.162
     1819498.588      255519.723     1819249.595      255827.798
#Sta/Elev= 30
       0 1607.58      20 1602.02      55 1590.48    94.9 1575.22   109.9 1567.91
   134.9 1558.22   184.8 1541.06   229.8 1520.16   264.7 1500.33   274.7 1497.84
   299.7 1494.05   324.7 1485.28   349.4 1482.03   371.8 1475.28   379.1 1474.25
   386.8 1474.85   413.6 1478.35     463 1479.72   497.6 1482.42   507.4 1484.19
   556.8 1502.43   670.7 1539.36   715.3 1558.41     745  1573.4   774.7  1586.6
   809.4 1604.05   839.1 1620.81   863.8 1636.71   913.3 1665.67     948  1684.3
#Mann= 3 , 0 , 0
       0      .1       0   371.8    .045       0   386.8      .1       0
Bank Sta=371.8,386.8
XS Rating Curve= 0 ,0
Exp/Cntr=0.3,0.1

Type RM Length L Ch R = 1 ,3999    ,540.8,543.2,545.7
XS GIS Cut Line= 4
     1819140.738      254926.359     1819127.209      255306.602
     1819078.677      255452.199     1819097.433      255863.682
#Sta/Elev= 30
       0 1569.54    19.8  1559.7    54.4 1549.42      84  1537.9   123.5 1530.07
   143.3  1525.2   202.6 1515.09     252 1499.61   286.6 1493.59   331.1 1482.49
   370.6 1474.46   400.3  1471.2     430 1470.03   466.5 1464.63   474.6 1463.79
   481.5 1464.93   499.3 1468.55   514.2 1473.23   568.7 1499.68   613.4  1518.6
   653.1 1534.16   697.7 1553.53   707.6 1558.77   737.4 1577.07   757.3 1585.79
     802  1608.1   831.7 1621.18   871.4 1646.89   896.2 1661.94   945.9  1687.9
#Mann= 3 , 0 , 0
       0      .1       0   466.5    .045       0   481.5      .1       0
Bank Sta=466.5,481.5
XS Rating Curve= 0 ,0
Exp/Cntr=0.3,0.1

Type RM Length L Ch R = 1 ,3455.8  ,311.5,309.9,308.3
XS GIS Cut Line= 3
     1819005.777      254884.736     1818639.775      255144.124
     1818415.563      255597.725
#Sta/Elev= 30
       0 1664.78      10 1666.49    34.9 1667.47    59.8 1665.92    89.7 1657.46
   104.7 1651.55   134.6 1637.62   159.5 1623.55   199.4 1603.08   224.3 1587.75
   254.2 1572.48     304 1543.86   338.9 1522.04   358.9 1512.84   398.8 1491.81
   468.4 1461.01   487.3 1453.91   488.3 1453.67   502.3 1455.41   537.9 1456.41
   607.3 1460.07   627.2 1463.99   666.9 1475.36   726.4 1496.68   761.1 1511.46
   810.7 1535.94   885.1 1571.22   909.9 1582.64   934.7 1592.21   954.6 1601.01
#Mann= 3 , 0 , 0
       0      .1       0   487.3    .045       0   502.3      .1       0
Bank Sta=487.3,502.3
XS Rating Curve= 0 ,0
Exp/Cntr=0.3,0.1

Type RM Length L Ch R = 1 ,3145.9  ,225.5,221.6,217.7
XS GIS Cut Line= 4
     1818475.519      254622.308     1818357.021      255009.077
     1818310.598      255123.023     1818051.055      255397.337
#Sta/Elev= 30
       0 1628.33      20 1618.68      45 1608.85    59.9 1602.25   109.9 1577.85
   199.8 1539.22   219.7  1527.8   244.7 1512.14   264.7 1502.63   269.7 1500.95
   274.7 1500.27   309.6  1499.8   314.6 1499.24   344.6 1489.37   354.6  1485.5
   369.6  1475.5   379.5 1469.79   404.5 1459.93   414.4 1455.34   429.1 1452.83
   448.8 1446.68   449.9 1446.68   453.7  1446.7   464.9 1448.46   478.3 1450.02
   671.6 1453.05   785.9 1456.96   830.7 1456.54   880.4 1458.08   905.2 1457.82
#Mann= 3 , 0 , 0
       0      .1       0   449.9    .045       0   464.9      .1       0
Bank Sta=449.9,464.9
XS Rating Curve= 0 ,0
Exp/Cntr=0.3,0.1

Type RM Length L Ch R = 1 ,2924.3  ,128.4,151.3,174.4
XS GIS Cut Line= 4
     1818363.351      254515.313      1818139.68      254939.444
     1818118.579      255036.509     1818036.285      255357.244
#Sta/Elev= 30
       0 1614.92      30 1598.31    89.9 1563.93    99.9 1558.57   109.9 1554.09
   139.8 1537.04   189.8 1512.97   224.8 1500.22   244.7  1494.8   294.7 1485.48
   309.7  1480.5   324.7 1473.46   344.6 1466.48   379.6 1455.84   404.6 1449.63
   414.6 1448.67   439.5  1447.9   489.4 1447.69   499.4 1446.89   510.8 1444.74
   519.2 1443.36   525.8 1443.89   544.1 1448.03     554 1448.72   598.6 1449.45
   613.4  1450.5   707.3  1453.4   746.9 1453.16   786.4 1453.75     910 1457.28
#Mann= 3 , 0 , 0
       0      .1       0   510.8    .045       0   525.8      .1       0
Bank Sta=510.8,525.8
XS Rating Curve= 0 ,0
Exp/Cntr=0.3,0.1

Type RM Length L Ch R = 1 ,2773    ,215.6,211,206.3
XS GIS Cut Line= 4
     1818310.598      254502.652     1818112.249      254852.929
     1817920.229      254920.453     1817823.164      255173.665
#Sta/Elev= 30
       0  1598.1    34.8 1575.92    69.6  1557.5   124.2 1525.41   144.1 1516.49
   178.9  1504.4   203.8 1492.67   233.6 1476.82   268.4  1472.4   298.2 1467.24
   377.7 1447.95   422.4 1447.42   457.2 1444.58   484.4 1439.95   486.9 1439.59
   499.4 1441.64   526.6 1447.55   546.5 1449.15   556.4 1449.68   576.3 1447.82
   606.1 1447.46   625.8 1447.98   635.7 1449.69   675.1  1476.1   704.7 1492.54
   734.3 1512.17   744.1 1517.82   768.8 1535.12     828 1573.34   877.3 1602.36
#Mann= 3 , 0 , 0
       0      .1       0   484.4    .045       0   499.4      .1       0
Bank Sta=484.4,499.4
XS Rating Curve= 0 ,0
Exp/Cntr=0.3,0.1

Type RM Length L Ch R = 1 ,2562    ,174.4,168.3,162.1
XS GIS Cut Line= 4
     1818298.066      254416.591     1817996.193       254660.91
     1817882.247      254730.543     1817557.422      254946.172
#Sta/Elev= 30
       0 1626.74      10 1619.85    74.7 1582.58    99.6  1565.4   124.5 1550.47
   159.3 1525.49   184.2 1509.38   219.1 1489.98   258.9 1471.08   288.8 1465.69
   328.6 1451.33   378.4 1445.58     423 1444.19   447.9 1438.41   457.6 1437.41
   462.9 1437.79   497.2  1444.3   531.9 1448.48   551.9 1453.42   586.9 1459.08
   621.9 1467.44   661.8 1472.75   731.8 1490.95   776.8 1497.03   796.8 1503.48
   816.8 1507.21   846.8 1516.68   861.8 1518.74   876.8 1518.01   911.8 1526.99
#Mann= 3 , 0 , 0
       0      .1       0   447.9    .045       0   462.9      .1       0
Bank Sta=447.9,462.9
XS Rating Curve= 0 ,0
Exp/Cntr=0.3,0.1

Type RM Length L Ch R = 1 ,2393.8  ,292.1,286.3,280.4
XS GIS Cut Line= 4
     1818122.799      254310.632     1817856.926      254538.524
     1817802.063      254597.607     1817441.235      254814.947
#Sta/Elev= 30
       0 1598.64    29.6 1577.06    64.1 1555.06   103.6 1523.19   133.2 1502.88
   162.8 1489.23   197.3 1470.05   221.9 1456.99   231.8 1452.48   241.7 1449.54
   276.2 1443.08   300.9 1440.97   335.4  1441.8   369.2 1438.11   384.2 1435.35
   388.1  1434.7   399.2 1436.49   421.3 1442.07   450.6 1456.76   470.4 1464.98
   485.3 1467.26   510.1 1468.08   544.8 1477.44   594.3 1492.68   624.1 1499.78
   668.7 1508.19   693.4 1514.04   703.4 1517.25   787.6  1550.3     852 1580.95
#Mann= 3 , 0 , 0
       0      .1       0   384.2    .045       0   399.2      .1       0
Bank Sta=384.2,399.2
XS Rating Curve= 0 ,0
Exp/Cntr=0.3,0.1

Type RM Length L Ch R = 1 ,2107.5  ,294.1,308.1,322.2
XS GIS Cut Line= 4
     1817829.011      253937.146     1817675.457      254295.861
     1817610.043      254418.248     1817351.278      254716.671
#Sta/Elev= 30
       0  1546.2    74.1 1514.16    93.8 1507.65   108.7 1505.92   148.2 1508.41
   172.9 1506.62   197.6 1501.66   261.8 1483.68   271.7 1480.06   286.5 1471.57
   316.1 1449.85     321  1447.5   330.9 1444.65   355.6 1439.38     415 1437.25
   444.7  1431.7   446.3 1431.73   461.3 1432.77   509.2 1437.25   514.1 1438.54
     554 1455.94     609  1474.8     649 1489.56     749 1528.49     769  1536.8
     814 1559.69     824 1566.15     854 1582.78     914  1619.6     924 1624.76
#Mann= 3 , 0 , 0
       0      .1       0   446.3    .045       0   461.3      .1       0
Bank Sta=446.3,461.3
XS Rating Curve= 0 ,0
Exp/Cntr=0.3,0.1

Type RM Length L Ch R = 1 ,1799.4  ,255.2,255.1,254.9
XS GIS Cut Line= 4
     1817757.341      253915.338     1817442.935       254151.67
     1817249.215      254247.329     1817238.255      254624.333
#Sta/Elev= 30
       0  1553.6    34.8 1538.88    59.8 1530.68    84.6 1520.32     224 1476.07
   263.9 1466.71   323.6 1455.78   353.5 1441.66   363.4 1437.88     408 1435.16
   432.7  1429.3   442.4 1428.52   447.7 1429.19   471.9 1432.63   496.4 1431.55
     521  1434.1   599.6 1434.41   619.3 1436.76   629.2  1439.7   639.2 1445.03
     659 1458.53   673.9 1469.46   708.6 1497.58   718.6 1503.88   743.4 1515.89
   768.2 1526.75   912.1 1604.83     932 1614.17   971.6 1635.23   986.5 1640.66
#Mann= 3 , 0 , 0
       0      .1       0   432.7    .045       0   447.7      .1       0
Bank Sta=432.7,447.7
XS Rating Curve= 0 ,0
Exp/Cntr=0.3,0.1

Type RM Length L Ch R = 1 ,1544.3  ,356.3,330,303.7
XS GIS Cut Line= 4
     1817711.305      253812.235     1817325.179      253926.593
     1817160.591      254008.887     1816988.541       254377.78
#Sta/Elev= 30
       0 1629.34    39.8 1620.75    64.6 1611.08   144.2 1559.48     169 1544.32
   188.9  1534.3   218.8 1521.07   273.4  1492.5   323.2 1469.06   338.1 1460.34
   372.9 1437.41   382.8 1434.44   432.6 1431.39   441.2 1428.94   452.4 1427.73
   456.2 1428.07   477.3 1430.04   661.2 1430.18   700.9 1432.84   705.8 1434.87
   720.8    1444   745.6 1461.62   755.5 1465.35   780.3 1470.49   790.2 1475.12
     825  1498.1   859.7 1519.55   909.4 1557.42   934.2 1565.89   993.8 1583.62
#Mann= 3 , 0 , 0
       0      .1       0   441.2    .045       0   456.2      .1       0
Bank Sta=441.2,456.2
XS Rating Curve= 0 ,0
Exp/Cntr=0.3,0.1

Type RM Length L Ch R = 1 ,1214.3  ,142,135.1,128
XS GIS Cut Line= 5
     1817040.315      253494.021     1816998.113      253728.243
     1817002.333      253844.299     1817014.994      254139.714
     1816930.589      254287.421
#Sta/Elev= 30
       0  1485.2       5 1483.26    44.6 1471.79    84.3 1462.89    94.2 1459.52
   128.9  1445.5   188.4 1441.52   198.3    1440   242.8 1429.66   252.5 1428.93
   281.5  1428.6   311.4 1423.58   315.4 1423.46   326.4 1424.14   354.1 1428.06
   442.8 1428.56   472.4 1428.17   541.4 1429.36   580.8 1435.44   595.6 1439.49
   615.3 1443.51   649.8 1457.08   669.2 1467.47   674.1 1471.15     713 1505.24
   737.3 1523.02   756.8 1539.44   790.8 1566.29   805.4 1576.86   819.9 1586.53
#Mann= 3 , 0 , 0
       0      .1       0   311.4    .045       0   326.4      .1       0
Bank Sta=311.4,326.4
XS Rating Curve= 0 ,0
Exp/Cntr=0.3,0.1

Type RM Length L Ch R = 1 ,1079.3  ,410.1,426.8,443.4
XS GIS Cut Line= 4
     1816815.042      253366.356     1816854.626      253770.445
     1816928.479      253941.364     1816868.437      254329.333
#Sta/Elev= 30
       0 1478.64    79.2  1449.4      99  1443.8   113.9 1441.36   163.4 1439.51
   242.6 1427.84   277.3 1428.24   341.6 1426.46   415.8 1426.46     461  1421.6
   464.8 1421.51     476 1422.31   489.3 1424.56   567.7 1425.74   592.2 1426.67
   602.2 1428.29     627 1437.34   656.8 1445.24   666.8 1449.17   691.6  1462.9
   726.4 1471.97   741.3 1482.81   766.2 1489.78     786 1496.42   840.7 1531.43
   865.5 1548.92   885.4 1564.13   940.1 1602.49     960 1618.66   984.8 1644.22
#Mann= 3 , 0 , 0
       0      .1       0     461    .045       0     476      .1       0
Bank Sta=461,476
XS Rating Curve= 0 ,0
Exp/Cntr=0.3,0.1

Type RM Length L Ch R = 1 ,652.5   ,514.1,492,472.7
XS GIS Cut Line= 4
     1816664.187      253325.681      1816552.88       253664.94
     1816487.467      253821.088     1816396.533      254204.826
#Sta/Elev= 30
       0 1444.83    19.8 1436.82    24.8 1435.18    29.8 1434.41    99.2 1430.99
     119 1428.87   138.8 1425.28   188.4 1426.47   322.3  1425.3   386.9 1422.32
   406.8 1422.58   436.7 1420.12   446.4 1417.86   461.4  1416.6   486.5 1420.93
   536.3 1421.97   541.3 1423.47   546.3 1427.16   556.3  1437.2   566.3 1448.61
   586.2 1473.52   601.2 1490.56   621.2 1504.46   636.2 1516.16   656.1 1530.27
   691.1 1552.99     716 1568.09   825.9 1627.26   890.8 1659.17   920.7 1672.15
#Mann= 3 , 0 , 0
       0      .1       0   446.4    .045       0   461.4      .1       0
Bank Sta=446.4,461.4
XS Rating Curve= 0 ,0
Exp/Cntr=0.3,0.1

Type RM Length L Ch R = 1 ,160.5   ,107,119.7,126.6
XS GIS Cut Line= 4
     1816505.885      253050.066     1816052.786      253755.674
     1816099.208       253856.96     1816263.796      254217.788
#Sta/Elev= 30
       0 1475.95    44.9 1463.34    99.8  1453.2   144.8 1440.66   189.7 1436.62
   214.6 1432.76   249.6 1430.03   289.5 1427.63   329.4 1427.22   354.4 1425.04
   379.4 1425.25     599 1419.28   833.6  1419.5   882.2  1410.1   884.1 1410.22
   891.8 1411.17   899.1 1413.98   906.4 1416.15   920.9 1417.03   930.6 1419.35
   969.8 1439.87   984.7 1446.49  1019.4 1448.14  1034.2 1453.29  1054.1 1462.79
  1168.1 1538.55  1232.6 1576.18  1287.1 1613.64  1326.7 1639.28  1346.6 1654.34
#Mann= 3 , 0 , 0
       0      .1       0   884.1    .045       0   899.1      .1       0
Bank Sta=884.1,899.1
XS Rating Curve= 0 ,0
Exp/Cntr=0.3,0.1

Type RM Length L Ch R = 1 ,40.8    ,27.3,23,24.3
XS GIS Cut Line= 4
     1816417.971      253016.938     1815953.611      253791.546
     1815970.491      253926.593      1816164.51        254255.8
#Sta/Elev= 30
       0 1451.88    39.9 1440.46    54.9 1438.12   219.6 1427.26   249.5 1427.82
   279.4 1425.47   329.3 1425.32   349.3 1424.06   434.1 1424.59     504 1422.89
   603.8 1423.35   808.3 1420.91   868.2  1418.3   910.5 1409.98   917.7 1409.41
   925.5 1409.58   946.9 1410.93   980.9 1418.01  1024.6 1420.35  1029.5  1421.4
  1088.9 1443.47  1128.6 1461.24  1148.4 1474.19    1203 1516.37  1212.9 1523.13
  1257.6 1552.54  1322.1 1592.92  1366.8 1623.05  1391.6 1642.13  1421.4 1667.41
#Mann= 3 , 0 , 0
       0      .1       0   910.5    .045       0   925.5      .1       0
Bank Sta=910.5,925.5
XS Rating Curve= 0 ,0
Exp/Cntr=0.3,0.1

Type RM Length L Ch R = 1 ,17.8    ,12.8,17.8,22.9
XS GIS Cut Line= 4
     1816011.527      253512.571     1815929.983      253761.024
      1815941.45      253934.304     1816169.517      254362.408
#Sta/Elev= 30
       0 1421.78    44.4 1421.02    78.9  1421.7   133.2 1421.47   182.6 1419.93
     222 1416.97   261.5 1409.87   276.4 1407.86   295.8 1407.19   306.2 1406.84
   310.8 1406.93   370.6 1409.21   380.6 1411.12   405.4 1417.59   440.1  1420.4
   474.8 1432.18   494.6  1440.5   504.4 1445.58   524.2 1457.47     549 1476.26
   578.7 1501.62   638.1 1546.49   672.7 1568.83   717.3 1594.76   766.8 1628.02
   796.5  1650.9   811.3 1663.14     846 1686.33   885.6 1716.92   920.2    1745
#Mann= 3 , 0 , 0
       0      .1       0   295.8    .045       0   310.8      .1       0
Bank Sta=295.8,310.8
XS Rating Curve= 0 ,0
Exp/Cntr=0.3,0.1

Chan Stop Cuts=-1
Use User Specified Reach Order=0
